--- MntnCrk.prj (project) ---

Proj Title=MntnCrk
Current Plan=p01
Default Exp/Contr=0,0
English Units
Geom File=g01
Flow File=f01
Plan File=p01
BEGIN DESCRIPTION:
END DESCRIPTION:
DSS Export Rating Curves= 0
DSS Export Rating Curve Sorted= 0
DSS Export Volume Flow Curves= 0
DXF OffsetX= 0
DXF OffsetY= 0
DXF ScaleX= 0
DXF ScaleY= 0

--- MntnCrk.p01 (plan) ---

Plan Title=Floodplain
Program Version=4.00
Geom File=g01
Flow File=f01
K Sum by GR=0
Std Step Tol=0.01
Critical Tol=0.01
Num of Std Step Trials=20
Max Error Tol=0.3
Flow Tol Ratio=0.001
Split Flow NTrial=30
Split Flow Tol=0.02
Split Flow Ratio=0.02
Log Output Level=0
Friction Slope Method=1
Unsteady Friction Slope Method=2
Unsteady Bridges Friction Slope Method=1
Global Log Level=0
CheckData=False
Run HTab=0
Run UNet=0
Run PostProcess=0
UNET Theta=0
UNET Theta Warmup=0
UNET ZTol=0
UNET ZSATol=0
UNET MxIter=0
UNET MaxInSteps=0
UNET DtIC=0
UNET DtMin=0
UNET MaxCRTS=0
UNET WFStab=0
UNET SFStab=0
UNET WFX=0
UNET SFX=0
UNET DSS MLevel=0
UNET DZMax Abort=0
UNET Convert EG Bridges=0
UNET Use Existing IB Tables=0
UNET Froude Limit=0
UNET Froude Power=0
Write IC File=0
Echo Input=False
Echo Output=False
Write Detailed=0

--- MntnCrk.f01 (steady flow) ---

Flow Title=NFF Regression Equation
Program Version=4.00
Number of Profiles=1
Profile Names=P100yr
River Rch & RM=MntnCrk,Main      ,39224.8
304.1069
River Rch & RM=MntnCrk,Main      ,38919.2
517.1070
River Rch & RM=MntnCrk,Main      ,36433.6
572.2386
River Rch & RM=MntnCrk,Main      ,35225.3
633.9459
River Rch & RM=MntnCrk,Main      ,30808.1
701.8601
River Rch & RM=MntnCrk,Main      ,30469.4
792.4283
River Rch & RM=MntnCrk,Main      ,29301.1
856.8538
River Rch & RM=MntnCrk,Main      ,27296.8
903.9352
River Rch & RM=MntnCrk,Main      ,26895.4
1166.639
River Rch & RM=MntnCrk,Main      ,25695.3
1210.317
River Rch & RM=MntnCrk,Main      ,20890
1340.717
River Rch & RM=MntnCrk,Main      ,20513
1769.767
River Rch & RM=MntnCrk,Main      ,14151.6
1878.439
River Rch & RM=MntnCrk,Main      ,13743.3
2988.318
River Rch & RM=MntnCrk,Main      ,6908.4
3227.440
River Rch & RM=MntnCrk,Main      ,506.9
3580.010
Boundary for River Rch & Prof#=MntnCrk,Main      ,1
Up Type=0
Dn Type=3
Dn Slope=0.028909

--- MntnCrk.g01 (geometry) ---

Geom Title=USGS 3m DEM
Program Version=4.10

River Reach=MntnCrk         ,Main
Reach XY= 30
     1937107.518      207125.473     1937252.217      204446.682
     1937037.033      203302.255     1937711.501      201325.527
     1939610.437      199905.536     1940543.957      199747.974
     1942117.975      198314.889      1944023.77      198316.645
     1944562.246      197742.481     1945541.009      197685.186
     1946411.404      196898.057     1946796.345      197411.571
     1948119.669      197908.965     1948688.223      197620.134
     1949010.881      197936.287     1949802.532      197846.622
     1951367.334      198262.232     1952296.731       197898.38
     1953618.157      198106.719     1954954.598       197412.97
     1955507.154      195365.013      1956719.43       195087.48
     1957372.732      195606.487     1957499.274      195014.645
     1958280.027      195064.435     1958739.691      195409.885
      1959470.43      194913.624     1960311.907      196120.848
     1961737.285      194695.181     1962927.714      194653.317

Type RM Length L Ch R = 1 ,39224.8 ,304.1,305.3,306.6
XS GIS Cut Line= 3
     1937418.872      207084.945     1937267.294      207080.735
     1936706.245      207068.103
#Sta/Elev= 30
       0 2591.01      19 2580.66    28.4 2571.18    47.4 2561.13    66.3 2552.82
    94.8 2542.81   113.7 2534.06   132.7 2527.79   142.2 2524.96   171.3 2518.71
   181.2 2515.54   250.1 2505.24   259.9 2503.02   279.6 2501.74   289.5 2501.85
   358.4 2506.98   407.6 2508.76   486.4  2521.2   506.1 2526.72   535.6 2532.37
   545.4 2534.83   565.2 2541.31   584.8 2551.08   614.4  2560.3   643.9 2570.46
   653.8 2575.63   663.6 2581.92   693.1 2594.84     703 2597.99   712.8 2599.36
#Mann= 3 , 0 , 0
       0      .1       0   279.6    .045       0   289.5      .1       0
Bank Sta=279.6,289.5
XS Rating Curve= 0 ,0
Exp/Cntr=0.3,0.1

Type RM Length L Ch R = 1 ,38919.2 ,465.8,464.8,463.8
XS GIS Cut Line= 3
     1937471.447      206822.256      1936852.37      206791.376
     1936659.739      206789.271
#Sta/Elev= 30
       0 2729.89      10 2724.07      70 2697.34     150 2649.65     160 2638.85
     170 2631.09   229.9 2592.83   239.9 2581.32   249.9 2572.75   309.9 2529.74
   319.9 2517.22   329.9 2507.93   349.9  2494.2   359.9 2489.99   369.9 2488.43
   431.7 2485.35   439.9 2485.14   446.7 2485.52   469.9 2489.12   489.9  2494.8
   549.9 2503.85   629.5 2529.56   648.7 2540.27   706.5 2564.11   725.8 2577.06
   745.1  2585.9   754.7 2589.79   764.3 2590.42   802.9 2610.32   812.5 2620.67
#Mann= 3 , 0 , 0
       0      .1       0   431.7    .045       0   446.7      .1       0
Bank Sta=431.7,446.7
XS Rating Curve= 0 ,0
Exp/Cntr=0.3,0.1

Type RM Length L Ch R = 1 ,38454.5 ,417.5,415,413.3
XS GIS Cut Line= 2
     1937365.408      206358.757     1936670.646      206363.036
#Sta/Elev= 30
       0 2597.55    39.7 2577.79    49.6 2571.15    59.6 2562.87   119.1  2533.4
     129 2527.06     139 2518.48   168.7 2504.07   198.5 2488.28   208.4 2482.03
   218.4 2472.93   228.3 2468.25   238.2 2464.86   262.7 2460.76     268 2460.38
   277.7 2460.92   297.8 2463.58   357.3  2468.3   367.2 2469.88   377.2 2473.94
   446.6 2507.02   456.6 2516.27     526 2549.09     536 2558.55   605.4 2593.52
   615.4 2603.21   625.3 2608.81   645.2 2619.05   655.1 2619.63   694.8 2638.65
#Mann= 3 , 0 , 0
       0      .1       0   262.7    .045       0   277.7      .1       0
Bank Sta=262.7,277.7
XS Rating Curve= 0 ,0
Exp/Cntr=0.3,0.1

Type RM Length L Ch R = 1 ,38039.2 ,392.2,400,405.6
XS GIS Cut Line= 3
     1937498.804      205908.785     1937089.505      205956.368
     1936681.161      205986.818
#Sta/Elev= 30
       0  2608.6    29.4 2607.76    68.7 2603.34   107.9 2589.93   127.5 2579.92
   186.4  2559.3     206 2545.86   235.5 2530.25   264.9 2512.81   274.7 2504.45
   284.5 2493.46     363 2445.15   404.6 2439.08   412.1 2438.91   419.6 2439.39
     472 2448.59   511.9 2460.39   521.9 2466.01   531.9 2469.28   591.8 2487.38
   601.8 2493.54   661.7 2514.95   671.7 2522.04   741.6 2552.05   751.6 2559.78
   761.6 2564.74   781.6  2573.3   791.6 2574.15   801.6  2577.7   821.5  2586.7
#Mann= 3 , 0 , 0
       0      .1       0   404.6    .045       0   419.6      .1       0
Bank Sta=404.6,419.6
XS Rating Curve= 0 ,0
Exp/Cntr=0.3,0.1

Type RM Length L Ch R = 1 ,37639.2 ,402.1,402,403.7
XS GIS Cut Line= 3
     1937512.223      205658.711     1937114.306      205564.964
     1936707.596       205494.07
#Sta/Elev= 30
       0 2536.13    39.9 2526.24    59.8 2518.63   119.6 2506.14   129.6 2502.28
   139.6 2495.65   159.5 2485.83   189.4 2476.29   219.4 2463.79   289.2 2443.62
   299.1 2438.36   309.1 2435.76   368.9 2429.38   401.3  2423.3   408.8 2422.82
   416.3 2423.78   448.1 2431.94   467.8 2440.39   526.8 2459.35   536.6 2463.26
   546.4  2471.4   575.9 2485.82   615.2 2500.17   634.9 2509.68   693.9 2528.85
   713.5 2540.43   772.5 2554.22   792.2 2563.47     802 2566.37   821.6 2568.43
#Mann= 3 , 0 , 0
       0      .1       0   401.3    .045       0   416.3      .1       0
Bank Sta=401.3,416.3
XS Rating Curve= 0 ,0
Exp/Cntr=0.3,0.1

Type RM Length L Ch R = 1 ,37237.2 ,352,349.3,345.6
XS GIS Cut Line= 3
     1937531.248      205261.417     1937129.894      205171.725
     1936735.249      205062.483
#Sta/Elev= 30
       0 2581.02    29.4 2568.44      49 2558.01    58.8 2552.58    78.3 2536.85
   117.5 2515.31   146.9 2501.43   156.7 2494.41   225.2    2465     235 2457.42
   244.8 2452.02   303.5 2429.11   323.1 2419.73   389.9 2400.34   391.7 2399.76
   404.9 2403.18   421.2 2411.54   471.2 2429.47   491.2 2441.54   521.1 2454.81
   551.1  2470.3     571 2487.25     601 2504.37     641 2532.19     651 2544.44
   720.9 2588.02   730.8 2598.71   740.8 2606.57   800.8 2642.24   820.7 2659.12
#Mann= 3 , 0 , 0
       0      .1       0   389.9    .045       0   404.9      .1       0
Bank Sta=389.9,404.9
XS Rating Curve= 0 ,0
Exp/Cntr=0.3,0.1

Type RM Length L Ch R = 1 ,36888   ,461.9,454.2,452.8
XS GIS Cut Line= 3
     1937579.974      204969.566     1937297.487      204847.934
     1936785.596      204789.953
#Sta/Elev= 30
       0 2548.47    39.7 2529.42    59.5  2515.8     129 2480.12   148.8 2463.74
   178.6 2445.67   198.4  2438.7   218.3 2433.83   228.2 2428.06   238.1 2424.69
   307.6 2404.98   317.5 2399.43   327.4 2396.46   347.2  2392.7   417.1 2383.91
   426.4 2383.36   432.1 2383.84   446.3 2387.68   466.1 2397.82     476 2406.02
   545.3 2437.53   555.2  2446.1   565.1 2452.18   624.6 2484.01   644.4 2500.28
   703.8 2529.49   723.6 2544.36   783.1 2574.82   802.9  2587.7   822.7 2595.36
#Mann= 3 , 0 , 0
       0      .1       0   417.1    .045       0   432.1      .1       0
Bank Sta=417.1,432.1
XS Rating Curve= 0 ,0
Exp/Cntr=0.3,0.1

Type RM Length L Ch R = 1 ,36433.6 ,400,399.9,401.8
XS GIS Cut Line= 3
     1937644.474      204323.862      1937241.44      204398.947
     1936841.522      204489.555
#Sta/Elev= 30
       0  2543.4      30 2537.99      50 2531.29      90 2514.42     100  2509.9
     110 2503.84     120 2495.51     190 2462.18     200 2453.19     270 2420.53
     280 2411.04     350 2378.88     360 2372.71   402.5 2363.84     410 2363.07
   417.5 2363.87   429.5 2367.54   439.3 2374.33     449 2379.58   507.6 2399.38
   517.4 2403.35   527.1 2408.96   595.5 2431.83   605.2 2438.49   673.6 2467.54
   693.1 2481.13   732.2 2500.22   761.4 2516.18   771.2  2527.3     820 2555.71
#Mann= 3 , 0 , 0
       0      .1       0   402.5    .045       0   417.5      .1       0
Bank Sta=402.5,417.5
XS Rating Curve= 0 ,0
Exp/Cntr=0.3,0.1

Type RM Length L Ch R = 1 ,36033.6 ,414.4,410.6,405.4
XS GIS Cut Line= 3
     1937612.388      203925.659     1937210.634      204003.776
     1936803.928      204061.333
#Sta/Elev= 30
       0 2496.57      20 2485.02    79.9 2464.02    99.8 2452.97   159.7 2429.82
   169.7 2424.48   179.7 2417.75   249.6  2387.2   259.5 2379.55   289.5 2367.83
   319.4 2357.47   339.4 2351.79   401.8 2347.07   416.8 2345.41   419.1 2345.14
   438.6 2347.44     468 2354.19   487.5 2360.09   507.1 2371.96   565.8 2399.03
   575.5 2405.53   585.3 2413.96   614.7 2429.98   653.8 2453.43   663.6 2465.14
     732 2510.72   741.8 2521.96   751.6  2529.7   800.5 2561.07     820 2574.72
#Mann= 3 , 0 , 0
       0      .1       0   401.8    .045       0   416.8      .1       0
Bank Sta=401.8,416.8
XS Rating Curve= 0 ,0
Exp/Cntr=0.3,0.1

Type RM Length L Ch R = 1 ,35623   ,385.5,397.6,411.4
XS GIS Cut Line= 3
      1937487.83      203476.521     1937104.416      203620.303
     1936723.452      203770.693
#Sta/Elev= 30
       0 2527.45      40 2506.79    49.9 2497.48    59.9 2491.34   119.8 2461.07
   129.8  2454.7   139.8 2446.14   179.8 2426.54   209.7 2413.22   219.7 2405.02
   229.7 2398.61   299.6 2356.97   309.6 2348.76   319.6 2345.65   359.6  2338.8
   379.5 2333.34   389.5 2328.78   399.5 2326.46   401.6 2326.53   416.6 2327.58
   469.4 2333.88   529.4 2343.29   549.3 2347.66   629.3 2374.17   639.2 2378.24
   649.2 2384.49   669.2 2392.43   709.2 2404.02   729.2 2407.19   819.1 2437.68
#Mann= 3 , 0 , 0
       0      .1       0   401.6    .045       0   416.6      .1       0
Bank Sta=401.6,416.6
XS Rating Curve= 0 ,0
Exp/Cntr=0.3,0.1

Type RM Length L Ch R = 1 ,35225.3 ,417.7,413.7,408.4
XS GIS Cut Line= 3
     1937457.087      203304.363     1937047.716      203231.926
     1936650.061      203138.857
#Sta/Elev= 30
       0 2530.87     9.9 2525.08    19.8 2515.91    49.5 2500.67    89.1 2477.26
      99 2465.38   168.3 2423.25   178.2 2413.84   188.1 2407.22   247.5 2377.23
   267.3 2362.69   316.8 2338.98   346.4 2322.86   366.2 2318.25   395.9 2309.25
   405.8 2307.56   408.2 2307.64   423.2 2309.27   535.3 2318.59   555.2 2323.38
   575.1 2331.44     595    2344   624.9  2357.3   654.8 2372.45   674.7 2388.83
   734.5 2426.67   744.4 2434.21   754.4  2445.8   764.4 2446.42   824.1 2485.18
#Mann= 3 , 0 , 0
       0      .1       0   408.2    .045       0   423.2      .1       0
Bank Sta=408.2,423.2
XS Rating Curve= 0 ,0
Exp/Cntr=0.3,0.1

Type RM Length L Ch R = 1 ,34811.5 ,366.8,375.1,384.9
XS GIS Cut Line= 3
     1937502.848      202832.405     1936969.479      202833.503
     1936678.727      202950.989
#Sta/Elev= 30
       0 2481.81    29.6 2463.59    59.3 2447.13      79  2432.4   138.3 2404.54
     158 2390.32   217.3 2361.95     237 2348.05   296.3 2319.26   306.2 2313.23
   316.1 2304.93   335.8 2296.29   345.7 2293.81     403 2287.76   414.8    2287
     418 2287.06   434.6 2288.64   464.2 2295.53   474.1 2299.97   493.9    2304
   562.8 2315.06   631.4 2328.74   690.2 2350.01   719.6 2363.96   729.4 2372.07
   739.2 2376.66     798 2398.76   817.6 2404.82   827.4 2411.55     847 2420.17
#Mann= 3 , 0 , 0
       0      .1       0     403    .045       0     418      .1       0
Bank Sta=403,418
XS Rating Curve= 0 ,0
Exp/Cntr=0.3,0.1

Type RM Length L Ch R = 1 ,34436.4 ,397.2,399.6,402.4
XS GIS Cut Line= 3
     1937558.111      202617.331     1937173.807      202472.997
     1936800.576      202304.943
#Sta/Elev= 30
       0 2452.06    39.1 2431.83    48.9 2423.86    58.6 2417.56   107.5 2394.37
   127.1 2387.18   136.8 2380.34   205.3 2351.81     215 2346.84   224.8 2339.94
   293.2 2309.51   312.8 2297.43   342.1 2286.17   371.4  2276.4     391 2271.59
   400.7 2270.77     403 2270.79     418 2271.23   470.4 2276.56   500.4  2281.1
   550.3 2295.68   560.3 2299.36   570.2 2304.98   640.1 2327.79   660.1 2337.76
     730 2365.75     750 2377.62   789.9 2393.28   809.8 2401.78   819.8 2406.92
#Mann= 3 , 0 , 0
       0      .1       0     403    .045       0     418      .1       0
Bank Sta=403,418
XS Rating Curve= 0 ,0
Exp/Cntr=0.3,0.1

Type RM Length L Ch R = 1 ,34035.5 ,339.4,339.5,337.8
XS GIS Cut Line= 3
     1937669.948      202287.628      1937301.35      202110.567
     1936947.672      201892.502
#Sta/Elev= 30
       0 2411.43      10 2402.15      20 2396.02    59.8  2376.3    89.8 2363.08
    99.7 2355.79   159.6 2331.16   179.5 2319.98   189.5 2311.12   199.5 2305.98
   229.4 2295.79   259.3 2283.83   269.3 2279.65   279.3 2273.96   299.2 2266.76
   309.2 2264.76   396.3 2256.64     399 2256.63   411.3 2259.23   428.7 2265.18
   448.5 2270.25   458.4 2276.55   537.5 2308.16   557.3 2319.26   636.5 2349.56
   646.4 2356.57   685.9 2374.58   725.5 2394.19   745.3 2408.81   824.4 2453.22
#Mann= 3 , 0 , 0
       0      .1       0   396.3    .045       0   411.3      .1       0
Bank Sta=396.3,411.3
XS Rating Curve= 0 ,0
Exp/Cntr=0.3,0.1

Type RM Length L Ch R = 1 ,33695.6 ,426.9,423.6,418.3
XS GIS Cut Line= 3
      1937872.04      202121.134     1937557.436      201862.946
     1937083.785      201634.122
#Sta/Elev= 30
       0 2402.28    19.8 2395.11    39.7 2391.12    69.5 2377.33   158.8 2343.18
   168.8 2338.11   208.5 2326.99   258.1 2308.05   277.9 2298.63   307.7 2288.69
   357.4 2276.31   387.1 2266.59   466.5 2248.83   506.2 2244.06   513.3 2244.19
   528.3 2245.49   615.4 2256.13   635.3  2267.1   655.1 2283.52   694.8 2304.63
   724.6 2315.78   744.4 2328.46   754.4 2332.54   784.1 2338.45   813.9 2341.96
   823.8 2345.23   873.5 2355.14   903.2 2362.03   913.2  2367.3     933 2372.82
#Mann= 3 , 0 , 0
       0      .1       0   513.3    .045       0   528.3      .1       0
Bank Sta=513.3,528.3
XS Rating Curve= 0 ,0
Exp/Cntr=0.3,0.1

Type RM Length L Ch R = 1 ,33271.2 ,440.8,454.4,467.9
XS GIS Cut Line= 3
     1938083.373      201611.311     1937887.238      201539.696
     1937204.717      201432.016
#Sta/Elev= 30
       0  2327.8    19.9 2322.43    89.5  2307.4   109.4 2301.43   129.3 2298.13
     179 2286.28   208.8 2276.86     268 2262.32   277.9 2257.84     347 2241.68
   356.9 2236.52   376.6 2229.46   386.5 2226.82   396.4 2225.94   406.2 2226.51
   465.4 2234.89   524.7 2240.91   554.3 2242.12     574 2244.91   583.9 2247.89
   593.8 2252.36   603.6 2259.05   672.7 2286.63   682.6 2294.33   712.2 2307.02
   751.7 2322.26   761.6 2328.42   781.3 2337.08   850.4 2358.31   899.8 2370.66
#Mann= 3 , 0 , 0
       0      .1       0   386.5    .045       0   406.2      .1       0
#XS Ineff= 2 , 0
          165.07 2290.58
Permanent Ineff=
       F       F
Bank Sta=386.5,406.2
XS Rating Curve= 0 ,0
Exp/Cntr=0.3,0.1

Type RM Length L Ch R = 1 ,32816.9 ,406.6,404.4,403.9
XS GIS Cut Line= 3
     1938218.141      201460.036     1937921.926      201177.287
     1937625.712      200894.537
#Sta/Elev= 30
       0 2340.29    59.9 2326.18    89.9 2317.14   109.9 2308.33   129.8 2302.14
   199.8 2284.19   209.7 2280.98   219.7  2276.2   249.7 2265.88   279.7 2254.25
   309.6 2240.23   329.6 2228.95   349.6 2226.08   369.6 2214.32   379.5 2210.22
   399.5 2210.96   459.4 2214.63   549.3 2218.43   569.3 2219.93   579.3 2222.14
   609.3 2239.72   619.2 2243.16   629.2 2248.27   659.2 2267.19   679.2 2284.05
   749.1 2325.23   759.1 2329.34   769.1 2331.88     789 2345.07     819 2360.69
#Mann= 3 , 0 , 0
       0      .1       0   379.5    .045       0   399.5      .1       0
Bank Sta=379.5,399.5
XS Rating Curve= 0 ,0
Exp/Cntr=0.3,0.1

Type RM Length L Ch R = 1 ,32412.5 ,404.1,412.3,418.8
XS GIS Cut Line= 3
     1938516.736      201140.327     1938194.232       200888.37
     1937890.157      200612.039
#Sta/Elev= 30
       0 2263.21      20 2261.16    79.9 2243.43   149.7 2224.13   169.7 2219.07
   179.7 2217.72   229.6  2204.3   239.6 2202.25   249.6 2201.39   329.4 2200.69
   401.8  2197.2   409.3 2196.99   416.8 2197.03   516.9 2204.01   526.6 2204.97
   536.4 2208.55   546.2 2214.24   575.6 2234.46   595.1 2253.54   614.7 2268.82
   624.5 2272.44   634.3 2277.16   663.6 2297.46   702.7 2319.96   712.5 2322.07
   741.9 2333.17   771.2 2340.36   800.6 2349.25   810.4  2352.9   820.1 2357.92
#Mann= 3 , 0 , 0
       0      .1       0   401.8    .045       0   416.8      .1       0
Bank Sta=401.8,416.8
XS Rating Curve= 0 ,0
Exp/Cntr=0.3,0.1

Type RM Length L Ch R = 1 ,32000   ,345.8,349.5,353.1
XS GIS Cut Line= 3
     1938752.634      200961.531     1938621.114      200832.326
     1938375.936      200431.427
#Sta/Elev= 30
       0 2269.28    19.4 2263.82    29.1 2261.82    48.5 2255.44    58.2 2251.89
    77.6 2241.69   116.4 2226.91   155.3 2210.62     165 2207.89   174.7 2205.95
   184.4 2201.89   194.4 2199.76   234.4 2194.55   264.4 2193.67   304.4 2193.24
   344.3 2191.79   384.3 2189.15   404.3 2188.44   444.3 2183.99   454.3 2184.33
   484.3 2186.88   524.3 2188.73   534.3 2189.86   544.3 2192.86   554.3 2197.06
   604.3 2220.07   614.3 2223.29   624.3 2225.84   644.3 2234.37   654.3 2235.41
#Mann= 3 , 0 , 0
       0      .1       0   444.3    .045       0   454.3      .1       0
Bank Sta=444.3,454.3
XS Rating Curve= 0 ,0
Exp/Cntr=0.3,0.1

Type RM Length L Ch R = 1 ,31650.7 ,471.8,458.5,445.2
XS GIS Cut Line= 2
     1938949.024      200894.153     1938707.257      200245.888
#Sta/Elev= 30
       0 2334.06    19.8  2324.4    29.6 2318.71    39.5 2314.51    49.4 2312.31
    59.3 2306.53    69.2 2300.11   108.7 2271.62   138.4 2251.47   148.3 2247.57
   158.1 2244.58   187.8 2227.48   227.3 2206.61   247.1 2194.78   276.8 2184.77
   286.6 2182.07   306.4 2178.79   316.3 2178.04   385.5 2175.63   395.4 2174.95
   415.1 2172.64   424.2 2172.28     425 2172.25   439.2 2173.23   454.7 2174.06
   563.4 2177.07   602.9  2183.8   612.8 2185.06   622.7 2185.28   691.9 2184.32
#Mann= 3 , 0 , 0
       0      .1       0   424.2    .045       0   439.2      .1       0
Bank Sta=424.2,439.2
XS Rating Curve= 0 ,0
Exp/Cntr=0.3,0.1

Type RM Length L Ch R = 1 ,31191.5 ,378.8,383.1,387.3
XS GIS Cut Line= 3
     1939451.072      200648.443     1939248.967      200330.375
      1938978.94      200138.209
#Sta/Elev= 30
       0  2305.5    59.5 2296.21    69.4 2295.46    79.3 2294.03    89.2 2290.34
   109.1 2286.43   128.9 2276.85   148.8 2265.62   178.5  2247.1   198.3 2233.45
   208.3 2231.32   218.2 2226.37   228.1 2218.37   247.9 2205.43   257.8 2199.67
   287.6 2184.25   317.4 2171.09   327.3 2170.08   347.1 2164.76     357 2162.77
   376.8 2160.14   492.4 2153.41   507.4 2152.59   513.3 2152.47   523.1 2152.66
   562.1 2155.89   620.5 2162.17   649.8 2164.23     679 2167.94   708.3 2170.43
#Mann= 3 , 0 , 0
       0      .1       0   492.4    .045       0   507.4      .1       0
Bank Sta=492.4,507.4
XS Rating Curve= 0 ,0
Exp/Cntr=0.3,0.1

Type RM Length L Ch R = 1 ,30808.1 ,323.3,338.7,354
XS GIS Cut Line= 3
      1939690.07      200369.986     1939537.216      200148.148
     1939156.197      199750.563
#Sta/Elev= 30
       0 2174.46    49.9 2162.52    59.9 2161.23   109.8 2161.83   129.7 2161.39
   189.6 2158.26   199.6 2157.44   219.5 2153.88   229.5 2153.36   249.4  2149.6
   269.4 2147.48   308.7 2145.24   367.7  2143.9   397.9 2142.14   407.1 2142.07
   412.9 2142.36   466.1  2144.6   515.2 2145.37   534.9 2147.55   554.6 2150.84
   584.1    2160   613.6 2171.92   623.4 2172.65   633.2 2175.75   682.4 2202.12
   751.2 2233.74   780.8  2237.7   790.6 2243.72   800.4 2250.96   820.1 2262.82
#Mann= 3 , 0 , 0
       0      .1       0   397.9    .045       0   412.9      .1       0
Bank Sta=397.9,412.9
XS Rating Curve= 0 ,0
Exp/Cntr=0.3,0.1

Type RM Length L Ch R = 1 ,30469.4 ,459.4,452.9,445.6
XS GIS Cut Line= 3
     1939767.484      200333.688     1939702.876      199729.027
     1939798.366      199478.909
#Sta/Elev= 30
       0 2181.79    39.9  2175.3    59.8 2173.71   139.6 2162.68   159.5 2161.38
   229.3 2148.46   249.2 2146.86   279.1 2142.67   434.3 2133.22   438.6 2133.12
   449.3 2133.26   458.6 2133.94   498.4 2140.61   508.4 2143.33   528.4 2153.16
   548.3 2154.01   568.2 2166.78   608.1 2194.61   637.8 2213.53   647.8 2214.22
   657.7 2218.65   727.1 2259.77     737  2264.8   746.9 2264.54   756.8 2270.56
   786.6 2291.42   836.2 2332.06   846.1 2337.38     856 2338.98   875.8 2353.63
#Mann= 3 , 0 , 0
       0      .1       0   434.3    .045       0   449.3      .1       0
Bank Sta=434.3,449.3
XS Rating Curve= 0 ,0
Exp/Cntr=0.3,0.1

Type RM Length L Ch R = 1 ,30016.4 ,419.8,419.8,420.1
XS GIS Cut Line= 3
     1940286.509      200179.518     1940117.321      199801.514
     1939909.174      199449.672
#Sta/Elev= 30
       0 2141.65    19.7 2138.07    39.4 2136.19    49.3 2135.93      69 2137.47
    88.7 2143.06    98.6 2144.59   118.3 2145.03     138 2141.52   167.6 2132.68
   177.5 2131.15   246.5 2127.41   315.5 2125.44   389.2 2121.08   394.4 2120.75
   404.2 2122.75   424.1 2125.17   434.1  2129.3   483.9  2155.8   533.8 2183.73
   543.8 2184.71   583.6 2209.06   633.5 2243.09   653.4 2249.51   683.4 2270.04
   703.3 2284.46   733.2 2304.42   753.2    2320   763.1 2320.93   822.9 2363.83
#Mann= 3 , 0 , 0
       0      .1       0   389.2    .045       0   404.2      .1       0
Bank Sta=389.2,404.2
XS Rating Curve= 0 ,0
Exp/Cntr=0.3,0.1

Type RM Length L Ch R = 1 ,29596.5 ,300.9,295,289.3
XS GIS Cut Line= 3
     1940696.839      200146.492     1940577.563      199851.616
     1940347.072      199337.396
#Sta/Elev= 30
       0 2254.26    19.9 2244.66    29.8 2243.17    59.6 2226.41    79.5 2212.82
    99.4 2195.74   109.3 2188.34   129.2 2178.74   139.2  2168.1   178.9 2144.64
   208.7 2128.77   238.6 2124.56   268.4 2123.63   367.5 2115.03   446.6 2110.14
   456.5 2109.67   466.4 2109.95   545.5 2116.38   555.4 2118.66   575.1 2126.53
   604.8 2142.96   624.6 2157.17   634.4 2159.79   644.3 2165.14   683.9 2195.91
   733.3 2226.66   753.1 2236.88   832.2 2286.75   851.9 2293.76   881.6 2312.29
#Mann= 3 , 0 , 0
       0      .1       0   446.6    .045       0   466.4      .1       0
Bank Sta=446.6,466.4
XS Rating Curve= 0 ,0
Exp/Cntr=0.3,0.1

Type RM Length L Ch R = 1 ,29301.1 ,395.2,386.9,377.4
XS GIS Cut Line= 3
      1940925.45       199844.99     1940786.295       199644.54
     1940517.756      199250.708
#Sta/Elev= 30
       0 2206.58    29.3 2190.46    48.8 2178.21    58.6 2174.64    68.3 2173.06
    97.6 2159.71   107.4 2156.34   117.1 2154.72   165.9 2131.12   185.4 2123.82
   224.5 2113.38   234.3 2112.27   263.9 2106.17   321.5 2103.95   336.5 2103.62
   363.2 2102.97   373.1 2103.43   412.8 2111.37   442.6 2123.06   452.6 2124.77
   472.4 2132.22   512.2 2156.86     532 2171.54   561.8 2195.44   581.7 2203.34
   631.3 2239.88     671 2266.63     681  2268.9   690.9  2272.9   720.7  2293.7
#Mann= 3 , 0 , 0
       0      .1       0   321.5    .045       0   336.5      .1       0
Bank Sta=321.5,336.5
XS Rating Curve= 0 ,0
Exp/Cntr=0.3,0.1

Type RM Length L Ch R = 1 ,28914.1 ,392.7,400,411.6
XS GIS Cut Line= 3
     1941332.024      199505.203     1940984.679      199289.209
     1940625.255      199089.004
#Sta/Elev= 30
       0 2244.86      20 2232.05    49.9 2215.44    59.9 2211.26    69.8 2209.77
    79.8 2205.14   119.7 2178.72   139.7 2164.28   179.6 2144.39   199.5 2135.73
   229.4 2126.19   319.2 2103.63   359.1 2097.11   401.5 2093.74     409 2093.52
   416.5 2093.75     507  2098.1   516.8 2101.65   536.4 2115.48   595.1 2163.36
   614.7  2183.8   683.3 2243.06   693.1 2252.64   702.9  2264.7   712.7 2271.39
   732.3 2282.11   761.7 2294.39   771.5 2297.21   800.8 2299.32   820.4  2302.8
#Mann= 3 , 0 , 0
       0      .1       0   401.5    .045       0   416.5      .1       0
Bank Sta=401.5,416.5
XS Rating Curve= 0 ,0
Exp/Cntr=0.3,0.1

Type RM Length L Ch R = 1 ,28514.1 ,394.4,402.3,403.8
XS GIS Cut Line= 3
     1941456.045      199276.379     1941187.697      198956.175
     1940972.272      198609.742
#Sta/Elev= 30
       0 2189.38    89.5 2138.82    99.5 2135.68   119.4 2131.86   169.1 2116.56
   318.3 2087.94   348.2 2085.97   410.3 2085.24   417.8 2085.23   425.3 2085.43
   527.2 2089.44   596.9 2090.67   606.8 2091.16   616.8  2094.6   626.7 2102.57
   646.6 2123.19   656.6 2132.42   666.5 2142.82   676.5 2154.58   686.4 2163.07
   696.4 2165.71   716.3 2179.04   746.1 2196.14   756.1 2203.79     776 2222.74
   785.9 2231.28   795.9 2238.58   805.8  2243.8   815.8 2247.76   825.7 2256.32
#Mann= 3 , 0 , 0
       0      .1       0   410.3    .045       0   425.3      .1       0
Bank Sta=410.3,425.3
XS Rating Curve= 0 ,0
Exp/Cntr=0.3,0.1

Type RM Length L Ch R = 1 ,28111.5 ,401.5,395.7,393
XS GIS Cut Line= 3
     1941687.958      199174.788      1941548.48      198793.812
     1941310.154      198435.225
#Sta/Elev= 30
       0 2266.03    29.7 2251.69    69.3 2228.88    79.2 2227.44    89.1 2221.62
   108.8 2208.55   138.5 2184.21   148.4 2177.05   168.2 2164.37   178.1 2159.28
     188 2157.32   217.7 2141.95   237.5 2134.04   267.2    2123     287 2118.58
   306.8 2111.12   326.5 2101.57   366.1 2079.34     376 2078.68   388.6 2075.87
   395.8 2074.98   403.6 2075.02   503.6 2077.82   669.9 2084.62   679.7 2086.47
   709.1 2099.77   728.6 2104.45   777.6 2125.24   826.5 2151.97   836.3 2158.56
#Mann= 3 , 0 , 0
       0      .1       0   388.6    .045       0   403.6      .1       0
Bank Sta=388.6,403.6
XS Rating Curve= 0 ,0
Exp/Cntr=0.3,0.1

Type RM Length L Ch R = 1 ,27715.7 ,417.9,418.6,419.3
XS GIS Cut Line= 3
     1942063.142      198866.219     1941887.937      198657.204
     1941513.545      198113.838
#Sta/Elev= 30
       0 2244.48     9.7 2240.37    48.7 2212.34    58.4 2210.58    68.2 2204.46
    87.7 2188.58   126.6 2154.46   146.1  2135.5   165.6 2119.99   175.3 2118.63
     224 2097.31   243.5  2089.9     263 2083.77   292.7 2075.92   302.7 2075.46
   322.7  2072.5   332.7 2071.89   447.9 2067.97   452.7 2067.86   462.9 2068.38
   502.7 2071.18   702.6 2079.87   762.6 2083.03   782.6 2087.14   812.6 2096.36
   852.6 2107.42   862.6 2112.24   872.6 2115.66   902.6 2123.48   932.6 2134.15
#Mann= 3 , 0 , 0
       0      .1       0   447.9    .045       0   462.9      .1       0
Bank Sta=447.9,462.9
XS Rating Curve= 0 ,0
Exp/Cntr=0.3,0.1

Type RM Length L Ch R = 1 ,27296.8 ,387,400.9,414.9
XS GIS Cut Line= 3
     1942350.029      198713.525     1942157.964      198368.955
     1941861.431      197928.299
#Sta/Elev= 30
       0 2154.43      69  2124.8    88.8 2121.17   118.4 2110.63   128.2 2108.27
   167.7 2102.19   187.4 2097.03   197.2  2096.3   256.4 2083.84     286 2079.84
   364.9 2074.04     424 2066.25   453.5 2059.78   463.3 2059.34   468.5 2059.67
   512.5 2066.44   532.2 2068.13   591.2 2079.84     660 2084.06   669.9 2083.16
   709.2  2085.1   768.2 2083.35   787.9 2087.24   807.6 2093.36   827.3 2101.83
   856.8 2117.62   866.6    2121   876.4 2118.32   896.1  2121.3   925.6 2128.09
#Mann= 3 , 0 , 0
       0      .1       0   453.5    .045       0   468.5      .1       0
Bank Sta=453.5,468.5
XS Rating Curve= 0 ,0
Exp/Cntr=0.3,0.1

Type RM Length L Ch R = 1 ,26895.4 ,387.7,396.6,400.3
XS GIS Cut Line= 3
     1942491.967      198696.735     1942502.072      198287.482
     1942533.839      197878.519
#Sta/Elev= 30
       0 2150.95    39.9 2134.65    49.9 2131.89    59.9 2130.87    89.9    2120
   139.8 2104.21   149.8 2101.67   159.8 2100.78   229.6 2075.89   380.2 2054.01
   389.4 2053.19   395.2  2054.2   399.4 2054.94   419.1 2065.06   428.9 2068.68
   438.7 2069.18   516.8  2103.4   526.6 2103.75   546.1 2107.16     634 2114.98
   643.8  2116.8   653.5 2121.18   682.8 2143.56   712.1 2167.72   721.9 2172.85
   731.7 2175.63     761 2200.12     800 2237.27   809.8 2245.52   819.6 2246.63
#Mann= 3 , 0 , 0
       0      .1       0   380.2    .045       0   395.2      .1       0
Bank Sta=380.2,395.2
XS Rating Curve= 0 ,0
Exp/Cntr=0.3,0.1

Type RM Length L Ch R = 1 ,26498.7 ,419,402.4,391.1
XS GIS Cut Line= 3
      1942722.88      198714.441     1942889.176      198341.663
     1942976.839      197926.495
#Sta/Elev= 30
       0  2143.7    49.8 2110.84    59.7 2106.04    69.7 2104.33    89.6 2103.64
   139.4 2099.48   159.3 2096.84   169.2 2094.26   179.2 2094.23   278.8  2060.6
   378.3 2050.42   427.9 2046.31   437.8 2045.56   447.7  2045.9   467.4 2052.47
   487.1    2056   566.1 2080.63   575.9 2083.07   585.8  2083.7   605.6  2089.9
   615.4 2090.22   674.6 2109.93   684.5 2110.58   694.4 2113.54   743.7 2131.89
   753.6 2135.74   763.4 2141.11   783.2 2147.99   812.8 2174.64   832.5  2194.5
#Mann= 3 , 0 , 0
       0      .1       0   427.9    .045       0   447.7      .1       0
Bank Sta=427.9,447.7
XS Rating Curve= 0 ,0
Exp/Cntr=0.3,0.1

Type RM Length L Ch R = 1 ,26096.3 ,388.3,400.9,413.3
XS GIS Cut Line= 3
     1943387.739      198691.292     1943271.189      198298.286
     1943159.583      197904.262
#Sta/Elev= 30
       0 2089.78      20  2086.3      60 2081.86      90 2077.52     160 2069.74
     230 2057.99   329.9 2048.97   349.9 2047.84   385.6 2043.52   389.9 2043.15
   400.6 2044.19   409.9 2048.02   419.9  2054.2   429.9 2058.43   439.9 2058.66
   529.8 2097.05   539.8 2098.66   549.8 2101.26   559.8 2105.46   579.7  2109.6
   609.7 2121.25   619.7 2124.26   639.7 2128.39   649.6 2129.01   729.6 2151.28
   739.5 2152.02   759.5 2157.79   769.5 2161.74   779.5 2168.16   819.4 2199.87
#Mann= 3 , 0 , 0
       0      .1       0   385.6    .045       0   400.6      .1       0
Bank Sta=385.6,400.6
XS Rating Curve= 0 ,0
Exp/Cntr=0.3,0.1

Type RM Length L Ch R = 1 ,25695.3 ,416.6,398.4,380.3
XS GIS Cut Line= 3
     1943558.103      198695.332     1943661.248      198299.036
     1943761.979      197902.109
#Sta/Elev= 30
       0 2133.43      30  2120.4      40 2117.52    49.9 2116.38   109.9 2088.72
   139.8 2078.74   149.8 2078.52   199.8 2063.99   229.7 2057.65   249.7 2055.75
   309.6 2046.07   339.6 2043.68   369.6 2039.66   379.5 2038.65   389.5 2038.95
   419.5 2050.37   429.5 2053.28   439.5 2053.44   499.4 2072.02   519.4 2077.02
   539.3 2079.67   559.3 2085.13   579.3 2088.29   629.2 2108.57   649.2 2112.33
   729.1  2145.8   739.1 2145.77   779.1 2161.96     789 2164.75     819 2167.32
#Mann= 3 , 0 , 0
       0      .1       0   369.6    .045       0   389.5      .1       0
Bank Sta=369.6,389.5
XS Rating Curve= 0 ,0
Exp/Cntr=0.3,0.1

Type RM Length L Ch R = 1 ,25296.9 ,407.7,397.6,387.5
XS GIS Cut Line= 3
     1944256.709       198650.54     1943981.885      198191.699
     1943899.922      197901.748
#Sta/Elev= 30
       0 2200.61    89.1  2147.1     109  2141.1   148.6 2118.16   158.5 2113.89
     208  2103.4   267.4 2094.08   287.2  2088.9     307  2075.9     317 2070.77
   326.8 2069.52   366.5 2047.97   386.3 2034.52   396.2 2029.14   399.5 2028.85
   406.1 2028.28   414.5    2030   435.8 2038.65   445.7 2040.16   485.3 2057.73
   505.1 2064.43   534.8 2070.79   593.2 2078.59   641.8 2087.25   651.5 2087.45
   680.6 2093.46     739 2116.64   758.4  2120.8   787.6 2131.26   836.2 2145.62
#Mann= 3 , 0 , 0
       0      .1       0   399.5    .045       0   414.5      .1       0
Bank Sta=399.5,414.5
XS Rating Curve= 0 ,0
Exp/Cntr=0.3,0.1

Type RM Length L Ch R = 1 ,24899.1 ,387.9,402.3,420.9
XS GIS Cut Line= 3
     1944673.122       198273.79     1944338.002      198037.264
     1943997.256      197810.364
#Sta/Elev= 30
       0 2145.11    19.5 2142.47    87.9  2137.7     166 2127.87   214.9 2116.43
   234.4 2113.79   283.2 2101.23   302.8 2093.97   312.5 2086.99   341.8 2074.17
   351.6 2068.37   390.6 2045.14   400.4 2037.18   410.2 2025.94   420.2 2021.66
   430.2 2021.19   434.5 2021.62   449.5 2024.06     510  2033.9   569.9 2039.51
   579.9 2041.57   589.9 2045.29   599.9 2052.39   659.8  2077.7   689.8  2088.5
   709.7  2100.8   749.7 2118.02   769.6 2125.15   789.6 2129.26   819.6 2138.91
#Mann= 3 , 0 , 0
       0      .1       0   434.5    .045       0   449.5      .1       0
Bank Sta=434.5,449.5
XS Rating Curve= 0 ,0
Exp/Cntr=0.3,0.1

Type RM Length L Ch R = 1 ,24496.2 ,382.4,386,386.4
XS GIS Cut Line= 3
     1944752.566      198196.292     1944586.963      197734.001
     1944522.603      197344.179
#Sta/Elev= 30
       0 2134.01    58.9 2128.26     108 2122.06   127.7 2120.69   137.5 2118.73
   157.1 2111.69   206.2 2089.15   216.1 2087.72   225.9 2084.74   314.3 2045.71
   324.1 2045.48   373.2 2026.69     383 2024.71   422.3 2021.78   483.6 2013.86
   491.1 2013.75   498.6 2015.42   520.7 2021.11   530.6 2026.34   599.7 2055.83
   609.6 2059.03   619.5 2060.07   639.2 2068.37   698.5 2087.15   708.4 2087.21
     738 2095.98   787.4 2105.27   807.1 2107.01   866.4 2115.69   886.2 2119.51
#Mann= 3 , 0 , 0
       0      .1       0   483.6    .045       0   498.6      .1       0
Bank Sta=483.6,498.6
XS Rating Curve= 0 ,0
Exp/Cntr=0.3,0.1

Type RM Length L Ch R = 1 ,24110   ,405.6,410.8,412.1
XS GIS Cut Line= 3
     1945071.974       198150.61     1944970.672      197750.524
     1944904.728      197345.906
#Sta/Elev= 30
       0 2122.16    19.6 2122.91    29.5 2121.98      59 2115.85    78.6 2113.65
   147.4 2090.05   157.2 2087.22     167 2087.19   245.7 2058.63   255.5 2057.63
   265.3 2055.26   343.9 2026.57   353.8 2024.44   363.6 2023.97   419.2 2009.85
   432.7 2008.45   434.2 2008.57   452.7 2009.48   502.7 2018.59   512.7 2021.32
   532.7 2029.96   542.7 2031.31   552.7  2034.8   632.7 2072.57   652.7 2077.54
   692.7  2096.7   702.7 2100.58   722.7 2104.41   742.7 2105.68   822.7 2114.81
#Mann= 3 , 0 , 0
       0      .1       0   419.2    .045       0   434.2      .1       0
Bank Sta=419.2,434.2
XS Rating Curve= 0 ,0
Exp/Cntr=0.3,0.1

Type RM Length L Ch R = 1 ,23699   ,396.3,380.5,367.7
XS GIS Cut Line= 3
     1945327.117      198078.693     1945352.266      197655.315
     1945323.145       197245.81
#Sta/Elev= 30
       0  2062.3    19.7  2058.9    78.9 2055.88    88.8    2056   108.5 2053.87
   118.4 2052.14   167.7 2039.75   177.5 2039.38   187.4 2037.59   256.4  2021.1
   276.2  2018.9   335.4  2006.7   355.1 2004.16   404.4  2002.4   416.6 2001.29
   431.6 1999.67   433.9 1999.46   453.4 2000.57   463.2 2002.17   482.8 2011.22
   512.1 2023.04   551.2 2041.36     561 2041.77   639.2 2077.71   648.9 2078.56
   678.3 2091.52   707.6 2101.21   727.1 2106.24   746.7 2108.17   834.7  2122.1
#Mann= 3 , 0 , 0
       0      .1       0   416.6    .045       0   431.6      .1       0
Bank Sta=416.6,431.6
XS Rating Curve= 0 ,0
Exp/Cntr=0.3,0.1

Type RM Length L Ch R = 1 ,23318.4 ,370.1,375,380
XS GIS Cut Line= 3
     1946025.443      197832.844     1945701.664      197601.482
     1945420.993      197218.307
#Sta/Elev= 30
       0 2080.53    29.8 2078.04    49.7  2074.9    79.6 2071.51   129.3 2063.09
   149.2 2056.97   179.1 2049.42     199  2045.7   238.8 2032.78   258.7 2024.09
   278.6 2018.18   298.5  2013.3   348.2 2003.05   368.1 2001.55   446.1 1988.91
   457.3 1988.33   461.1 1989.18   467.2 1990.54   477.1  1994.5     487  1996.7
   506.8 2003.97   595.8 2042.71   615.6 2047.57   665.1 2066.65   704.7 2079.93
   714.6 2082.06   724.5 2083.03   754.2 2091.48   823.4 2106.13   872.9 2113.77
#Mann= 3 , 0 , 0
       0      .1       0   446.1    .045       0   461.1      .1       0
Bank Sta=446.1,461.1
XS Rating Curve= 0 ,0
Exp/Cntr=0.3,0.1

Type RM Length L Ch R = 1 ,22943.3 ,347.7,337.8,328
XS GIS Cut Line= 3
     1946117.605      197772.603     1945974.844      197370.708
     1945805.773      196996.741
#Sta/Elev= 30
       0 2089.59    39.7 2086.62    99.2 2083.71     119 2081.24   148.8 2074.81
   168.6 2071.98   188.4 2064.55     248 2037.32   257.9 2036.69   287.6 2022.98
   337.2 2002.17   357.1 1997.97   386.8 1987.59   447.5 1977.82   455.8  1977.5
   462.5  1977.6   475.4 1979.39   494.9 1989.91   504.7 1993.29   563.3  2005.9
   592.6 2016.54   612.2 2022.18   651.2 2028.38   670.8  2029.4   680.6 2031.27
   729.4  2049.3   758.7 2056.58   768.5 2056.46   797.8 2066.34   836.9 2068.93
#Mann= 3 , 0 , 0
       0      .1       0   447.5    .045       0   462.5      .1       0
Bank Sta=447.5,462.5
XS Rating Curve= 0 ,0
Exp/Cntr=0.3,0.1

Type RM Length L Ch R = 1 ,22605.5 ,753.5,790.5,827.5
XS GIS Cut Line= 3
     1946370.698      197662.626      1946289.74      197205.835
     1945817.432      196801.261
#Sta/Elev= 30
       0 2088.39   118.4 2082.01   177.7 2080.72   236.9 2072.88   266.5 2064.18
   315.8 2042.78   335.6 2038.62   404.7 2006.57   434.3 1998.92   473.8 1980.65
   493.5 1974.89   517.9 1973.01   532.9 1972.72   542.9 1972.69   562.6 1973.92
   592.2 1979.47   631.7 1982.55   641.6 1985.19   671.2 2005.53     691 2013.46
   750.2 2054.55   809.4 2072.91   829.2 2075.43   898.2 2093.78     918 2097.76
   967.4 2104.19   977.2 2103.53  1026.6 2107.21  1066.1 2102.36  1085.8 2096.16
#Mann= 3 , 0 , 0
       0      .1       0   517.9    .045       0   532.9      .1       0
Bank Sta=517.9,532.9
XS Rating Curve= 0 ,0
Exp/Cntr=0.3,0.1

Type RM Length L Ch R = 1 ,21814.5 ,576.3,562.7,547.8
XS GIS Cut Line= 3
     1946412.394      197654.345       1946528.8      197303.256
      1947104.38      196715.221
#Sta/Elev= 30
       0 2092.99      30 2094.31     140 2091.94     160 2088.82   209.9  2075.6
   229.9 2072.38   309.9 2042.27   319.9 2041.32   339.9 2032.64   389.7  2002.6
   419.4 1974.35   429.4 1966.66   439.3 1961.26   465.6 1956.37   478.9 1956.15
   480.6  1956.2     697 1978.19   726.8 1982.79   766.4 2002.35   786.3 2017.15
     816 2034.31   835.8 2040.77   845.8 2045.86   915.1 2083.95   964.7  2107.1
   984.5 2121.67  1004.4 2132.78  1024.2 2141.38  1034.1 2143.52  1192.7 2151.95
#Mann= 3 , 0 , 0
       0     .06       0   465.6    .045       0   480.6     .06       0
Bank Sta=465.6,480.6
XS Rating Curve= 0 ,0
Exp/Cntr=0.3,0.1

Type RM Length L Ch R = 1 ,21251.5 ,348.6,361.3,375.5
XS GIS Cut Line= 3
     1947020.097      197880.257     1947066.482       197371.68
     1947120.884      197059.848
#Sta/Elev= 30
       0 2048.08    49.1 2014.98    58.9 2013.68    68.8 2008.59    98.2 1990.47
     108 1986.85   147.3 1976.57     167    1974   206.2 1964.74   343.7 1954.55
   373.2 1951.17   422.3 1942.83   437.3 1941.99   441.9 1941.95   471.4 1946.29
   560.2 1953.54     570 1955.55   579.9 1959.94   609.6 1977.08   629.4 1983.01
   678.8 2017.34   688.7 2025.36   708.5 2043.84   718.4 2050.74   728.3 2052.67
   738.2 2060.67   748.1 2066.79     758 2070.18   777.8 2073.24   827.2 2075.08
#Mann= 3 , 0 , 0
       0      .1       0   422.3    .045       0   437.3     .06       0
Bank Sta=422.3,437.3
XS Rating Curve= 0 ,0
Exp/Cntr=0.3,0.1

Type RM Length L Ch R = 1 ,20890   ,385.9,376.7,366.1
XS GIS Cut Line= 3
     1947132.618      197911.848     1947380.679      197583.433
     1947647.672      197273.384
#Sta/Elev= 30
       0 2046.68     9.8 2042.58      49 2020.28      98 1994.04   107.8 1991.05
   117.6 1989.54   166.6 1963.04   176.4  1958.8     196 1954.59   215.6 1951.52
   313.6 1943.48   372.4 1939.76   382.2 1938.83   404.1 1934.66   411.6 1933.91
   419.1  1934.4   421.6 1934.57   441.5 1941.16   451.5  1943.5   471.4 1945.88
   571.2 1965.67   591.2 1966.83   631.1 1976.82     681 1993.98     701 2002.72
     711 2005.84   720.9 2006.65   740.9 2016.81   800.8 2043.79   820.7 2054.44
#Mann= 3 , 0 , 0
       0      .1       0   404.1    .045       0   419.1      .1       0
Bank Sta=404.1,419.1
XS Rating Curve= 0 ,0
Exp/Cntr=0.3,0.1

Type RM Length L Ch R = 1 ,20513   ,786,770.9,755.6
XS GIS Cut Line= 3
     1947590.538        198160.5     1947698.471      197765.469
     1947803.751      197369.736
#Sta/Elev= 30
       0 1957.01    79.9 1953.97   159.8 1953.07   179.8 1952.24   229.7 1947.46
   239.7 1946.66   249.7 1946.75   259.7 1945.73   289.6 1941.26   329.6 1933.59
   339.6 1932.55   369.6 1931.52   431.7 1927.88   446.7 1927.47   449.5 1927.46
   459.4 1928.32   479.4 1934.63   549.3 1936.58   579.3 1938.48   609.3 1941.59
   629.2 1945.56   639.2 1946.57   649.2 1948.52   679.2 1959.51   719.1 1973.09
   729.1 1975.74   739.1 1976.73   779.1 1993.88     799 2004.55     819 2016.27
#Mann= 3 , 0 , 0
       0      .1       0   431.7    .045       0   446.7      .1       0
Bank Sta=431.7,446.7
XS Rating Curve= 0 ,0
Exp/Cntr=0.3,0.1

Type RM Length L Ch R = 1 ,19742   ,459.2,473,487
XS GIS Cut Line= 2
     1948487.193      198161.996     1948123.089      197304.372
#Sta/Elev= 30
       0 2092.08     9.9 2086.36    29.7 2081.08    39.6 2075.38    59.5 2070.99
   148.7 2012.84   158.6 2009.11   168.5 2007.63   198.2 1992.56   247.8 1970.96
   267.6 1967.78   346.9  1944.9   366.7 1942.65   426.2 1922.38   535.4 1912.62
   545.2 1912.38   550.4 1913.05     565 1914.57   624.4 1931.51   664.1 1945.07
     674  1946.1   693.8 1951.48   763.2 1962.98   773.1 1963.05   822.7 1970.42
   832.6 1973.43   862.3 1993.23   872.2 1994.74   892.1 2010.27   931.7 2037.76
#Mann= 3 , 0 , 0
       0      .1       0   535.4    .045       0   550.4      .1       0
Bank Sta=535.4,550.4
XS Rating Curve= 0 ,0
Exp/Cntr=0.3,0.1

Type RM Length L Ch R = 1 ,19268.9 ,383.4,390.2,396.8
XS GIS Cut Line= 3
     1948628.478      198148.899     1948729.084      197648.613
     1948829.212      197269.915
#Sta/Elev= 30
       0  2082.8     9.8  2082.6    29.4 2067.56    39.2  2067.2   117.8 2012.24
   137.4 2005.47   166.8 1985.64   215.9 1959.46   225.7 1955.03   235.5 1953.88
   294.4 1922.57     314 1914.24   343.5  1909.6   363.1 1908.84     471  1913.3
   490.7 1911.87   510.3 1906.24   523.7 1905.97   529.9 1905.92   538.7  1908.9
   559.3 1917.89   598.4  1927.2     618 1929.18   706.2 1943.59     716 1943.46
   735.5 1948.06   794.3 1969.56   813.9 1972.95   892.2 2003.98     902 2003.78
#Mann= 3 , 0 , 0
       0     .08       0   523.7    .045       0   538.7      .1       0
Bank Sta=523.7,538.7
XS Rating Curve= 0 ,0
Exp/Cntr=0.3,0.1

Type RM Length L Ch R = 1 ,18878.7 ,431,417.4,403.9
XS GIS Cut Line= 3
     1948698.712      198206.567     1948910.282      198039.291
     1949217.305      197523.789
#Sta/Elev= 30
       0 2101.93      10 2096.91      30 2084.68    59.9 2070.64    89.9 2054.67
   109.9 2049.91   139.8 2030.75   159.8 2025.56   219.8 1988.92   229.8 1981.83
   239.7  1976.5   279.6  1958.4   289.4 1957.24   299.2 1953.96     309 1948.71
   328.7 1935.23   338.6 1926.98   358.2 1907.67   368.1 1900.16   377.9 1895.09
   387.7 1893.26   405.9  1893.8   420.9 1894.92   476.3 1900.43   535.3  1900.9
   741.8 1912.57     791 1917.06   830.4  1922.7   840.2  1922.3   869.7 1927.43
#Mann= 3 , 0 , 0
       0     .08       0   405.9    .045       0   420.9     .08       0
Bank Sta=405.9,420.9
XS Rating Curve= 0 ,0
Exp/Cntr=0.3,0.1

Type RM Length L Ch R = 1 ,18461.3 ,338.3,343.4,350.9
XS GIS Cut Line= 3
      1949422.34      198384.982     1949390.833      197981.622
     1949366.716      197544.954
#Sta/Elev= 30
       0 2028.51    29.6 2019.38    49.3 2014.86    59.2 2013.02    78.9  2011.5
   108.6 2005.79   157.9 1988.34   167.8 1987.82   207.2 1971.27   236.8 1955.45
   246.7 1955.36   266.4 1944.96   276.3 1945.12   315.8  1922.7   335.5  1909.6
   355.2 1899.71   365.1 1899.19   394.7 1889.97   404.6 1887.85   413.8 1887.45
   414.5 1887.42   428.8 1888.28   543.7 1896.66   692.8 1897.62   702.8 1899.12
   732.6 1906.42   752.5 1909.69   782.3 1917.74     822 1926.99   841.9 1929.24
#Mann= 3 , 0 , 0
       0     .08       0   413.8    .045       0   428.8     .08       0
Bank Sta=413.8,428.8
XS Rating Curve= 0 ,0
Exp/Cntr=0.3,0.1

Type RM Length L Ch R = 1 ,18117.8 ,402.2,409.3,414.8
XS GIS Cut Line= 3
     1949652.441      198302.691     1949741.897      197737.789
     1949791.596      197512.491
#Sta/Elev= 30
       0 1976.13      69 1947.26    88.8 1943.26   147.9 1920.01   157.8 1917.35
   167.6 1916.35   177.5 1913.51   187.4  1912.7   256.4 1888.45   266.2 1885.93
   276.1 1884.99   364.9  1881.7     493 1877.64   502.9  1877.5   512.8 1878.95
   522.6  1883.2   532.5 1888.25   552.2 1896.57   562.1 1899.94   571.9 1900.81
   581.6 1905.06   591.2 1909.58   648.8 1940.23   658.5 1942.11   668.1  1945.4
   716.1 1972.33     745 1986.04   754.6 1991.19   764.2 1992.02   802.7 2011.62
#Mann= 3 , 0 , 0
       0      .1       0     493    .045       0   512.8      .1       0
Bank Sta=493,512.8
XS Rating Curve= 0 ,0
Exp/Cntr=0.3,0.1

Type RM Length L Ch R = 1 ,17708.4 ,407.7,399.9,391.8
XS GIS Cut Line= 3
     1949892.974      198322.384     1950079.856       197957.59
     1950280.584      197600.737
#Sta/Elev= 30
       0  1938.8      20 1933.59      70 1909.72      90 1902.15     100 1899.22
     120 1896.15     140 1890.28     170 1884.64   189.9  1881.9   229.9 1879.98
   269.9 1876.12   319.9  1872.5   402.4 1869.13   417.4 1868.36   419.9 1868.28
   429.8 1870.71   439.8 1871.21   469.8 1877.41   499.8 1888.06   529.7 1900.53
   549.7 1904.53   589.6  1923.9   639.6 1951.86   649.6 1956.35   659.5 1956.94
   699.5 1976.46   749.4 1999.13   759.4 2000.38   769.4 2003.22   819.3 2026.41
#Mann= 3 , 0 , 0
       0      .1       0   402.4    .045       0   417.4      .1       0
Bank Sta=402.4,417.4
XS Rating Curve= 0 ,0
Exp/Cntr=0.3,0.1

Type RM Length L Ch R = 1 ,17308.4 ,400.7,400,398.7
XS GIS Cut Line= 3
     1950386.711      198527.717     1950438.699      198121.555
     1950500.185       197716.56
#Sta/Elev= 30
       0  1923.7      20 1915.18      30 1914.26    89.9 1886.55    99.9 1882.47
   109.9 1879.58   119.8  1879.2   139.8 1875.82   199.7 1872.22   379.5 1863.12
   419.5  1862.2   439.4 1861.02   449.4 1860.32   459.4 1860.83   469.4  1865.8
   479.4 1873.81   489.4 1880.82   499.4 1882.85   509.4 1887.14   559.3  1918.8
   589.3 1939.58   609.3 1946.58   639.3 1966.04   679.2 1988.98   699.2 1994.38
   749.2 2019.47   769.2 2027.86   779.2 2030.66   789.1  2032.4   819.1 2043.86
#Mann= 3 , 0 , 0
       0      .1       0   439.4    .045       0   459.4      .1       0
Bank Sta=439.4,459.4
XS Rating Curve= 0 ,0
Exp/Cntr=0.3,0.1

Type RM Length L Ch R = 1 ,16908.4 ,345.7,343.9,342.1
XS GIS Cut Line= 3
     1950796.203      198578.328     1950835.557      198170.627
     1950873.669      197762.984
#Sta/Elev= 30
       0 1883.09      30 1878.02    59.9 1873.96    69.9 1873.86    99.9  1870.6
   159.8 1866.09   229.8 1863.05   289.7 1861.52   349.6 1858.64   429.6 1853.12
   459.5  1851.8   469.5 1851.26   479.5 1851.66   489.5 1855.01   509.4 1864.87
   529.4 1875.53   539.4 1881.63   549.4  1882.7   559.4 1888.01   579.4 1901.59
   599.3 1916.02   639.3 1947.68   649.3 1949.32   659.2 1954.96   689.2 1977.38
   699.2 1983.52   729.1  1998.3   739.1 1999.55   749.1 2001.96     819 2031.53
#Mann= 3 , 0 , 0
       0      .1       0   459.5    .045       0   479.5      .1       0
Bank Sta=459.5,479.5
XS Rating Curve= 0 ,0
Exp/Cntr=0.3,0.1

Type RM Length L Ch R = 1 ,16564.5 ,298.5,291.9,285.4
XS GIS Cut Line= 3
      1951160.42       198643.72     1951168.234      198363.985
     1951181.486      197765.951
#Sta/Elev= 30
       0 1882.01      30 1878.03      50 1876.45      80 1872.46   109.9 1869.88
   119.9 1869.14   139.9 1868.45   219.9 1863.55   239.9 1862.95   309.8 1858.38
   359.6 1857.34   369.6 1856.62   399.5 1852.36   419.4 1850.51   428.7 1849.27
   439.4 1848.88   449.3 1849.33   489.2 1851.36     569 1852.91   578.9 1854.95
   598.9 1862.45   618.8 1866.36   688.6 1894.14   698.6 1896.56   708.5 1898.28
   788.3 1931.22   798.3 1933.78   808.2 1935.33   838.2 1947.74     878 1964.83
#Mann= 3 , 0 , 0
       0      .1       0   428.7    .045       0   449.3      .1       0
Bank Sta=428.7,449.3
XS Rating Curve= 0 ,0
Exp/Cntr=0.3,0.1

Type RM Length L Ch R = 1 ,16272.5 ,572.2,564.1,558.9
XS GIS Cut Line= 3
     1951589.531       198628.78     1951486.394      198358.003
     1951341.699      197842.751
#Sta/Elev= 30
       0 1930.51      20 1925.09      30 1926.31      40 1922.98    69.9 1908.04
   109.9 1889.72   119.9 1886.43   129.9 1885.98   139.9 1881.43   159.9 1875.63
   169.9    1874   229.8 1873.02   239.8 1872.11   259.8 1868.65   319.5  1854.6
   329.4 1854.53     369 1845.64     379  1845.4   384.4 1845.72   408.7 1847.86
   448.3 1849.89   636.6 1852.65   646.5 1855.06   656.4 1859.11     706 1881.75
   715.9  1885.6   725.8 1886.51   765.5 1905.27     815 1927.28   824.9 1928.55
#Mann= 3 , 0 , 0
       0      .1       0     369    .045       0   384.4      .1       0
Bank Sta=369,384.4
XS Rating Curve= 0 ,0
Exp/Cntr=0.3,0.1
